--- macdonald.prj (project) ---

Proj Title=A1F-001 MacDonald backwater dx=5 m
Current Plan=p01
Default Exp/Contr=0,0
SI Units
Geom File=g01
Flow File=f01
Plan File=p01
Y Axis Title=Elevation
X Axis Title(PF)=Main Channel Distance
X Axis Title(XS)=Station
BEGIN DESCRIPTION:
A1F-001 MacDonald backwater dx=5 m
END DESCRIPTION:

--- macdonald.p01 (plan) ---

Plan Title=A1F-001 MacDonald backwater dx=5 m
Program Version=6.60
Short Identifier=dx5
Geom File=g01
Flow File=f01
Subcritical Flow
K Sum by GR= 0
Std Step Tol= .00001
Critical Tol= .00001
Num of Std Step Trials= 40
Max Error Tol= .3
Flow Tol Ratio= .001
Log Output Level= 0
Friction Slope Method= 1

--- macdonald.f01 (steady flow) ---

Flow Title=A1F-001 MacDonald backwater dx=5 m
Program Version=6.60
Number of Profiles= 1
Profile Names=PF 1
River Rch & RM=Channel,Main            ,1000
   20000
Boundary for River Rch & Prof#=Channel,Main            , 1
Up Type= 0
Dn Type= 1
Dn Known WS=0.690867

--- macdonald.g01 (geometry) ---

Geom Title=A1F-001 MacDonald backwater dx=5 m
Program Version=6.60

River Reach=Channel         ,Main
Reach XY= 2
          0.5000          1.0000          0.5000          0.0000

Type RM Length L Ch R = 1 ,1000    ,5,5,5
#Sta/Elev= 4
 0.00000       5 0.00000 0.00000  100000 0.00000  100000       5
#Mann= 3 ,0,0
 0.00000 0.03000 0.00000 0.00000 0.03000 0.00000  100000 0.03000 0.00000
Bank Sta=0,100000
XS Rating Curve= 0 ,0
Exp/Cntr=0,0

Type RM Length L Ch R = 1 ,995     ,5,5,5
#Sta/Elev= 4
 0.00000 4.99897 0.00000-0.00103  100000-0.00103  100000 4.99897
#Mann= 3 ,0,0
 0.00000 0.03000 0.00000 0.00000 0.03000 0.00000  100000 0.03000 0.00000
Bank Sta=0,100000
XS Rating Curve= 0 ,0
Exp/Cntr=0,0

Type RM Length L Ch R = 1 ,990     ,5,5,5
#Sta/Elev= 4
 0.00000  4.9979 0.00000-0.00210  100000-0.00210  100000  4.9979
#Mann= 3 ,0,0
 0.00000 0.03000 0.00000 0.00000 0.03000 0.00000  100000 0.03000 0.00000
Bank Sta=0,100000
XS Rating Curve= 0 ,0
Exp/Cntr=0,0

Type RM Length L Ch R = 1 ,985     ,5,5,5
#Sta/Elev= 4
 0.00000 4.99679 0.00000-0.00321  100000-0.00321  100000 4.99679
#Mann= 3 ,0,0
 0.00000 0.03000 0.00000 0.00000 0.03000 0.00000  100000 0.03000 0.00000
Bank Sta=0,100000
XS Rating Curve= 0 ,0
Exp/Cntr=0,0

Type RM Length L Ch R = 1 ,980     ,5,5,5
#Sta/Elev= 4
 0.00000 4.99564 0.00000-0.00436  100000-0.00436  100000 4.99564
#Mann= 3 ,0,0
 0.00000 0.03000 0.00000 0.00000 0.03000 0.00000  100000 0.03000 0.00000
Bank Sta=0,100000
XS Rating Curve= 0 ,0
Exp/Cntr=0,0

Type RM Length L Ch R = 1 ,975     ,5,5,5
#Sta/Elev= 4
 0.00000 4.99444 0.00000-0.00556  100000-0.00556  100000 4.99444
#Mann= 3 ,0,0
 0.00000 0.03000 0.00000 0.00000 0.03000 0.00000  100000 0.03000 0.00000
Bank Sta=0,100000
XS Rating Curve= 0 ,0
Exp/Cntr=0,0

Type RM Length L Ch R = 1 ,970     ,5,5,5
#Sta/Elev= 4
 0.00000  4.9932 0.00000-0.00680  100000-0.00680  100000  4.9932
#Mann= 3 ,0,0
 0.00000 0.03000 0.00000 0.00000 0.03000 0.00000  100000 0.03000 0.00000
Bank Sta=0,100000
XS Rating Curve= 0 ,0
Exp/Cntr=0,0

Type RM Length L Ch R = 1 ,965     ,5,5,5
#Sta/Elev= 4
 0.00000  4.9919 0.00000-0.00810  100000-0.00810  100000  4.9919
#Mann= 3 ,0,0
 0.00000 0.03000 0.00000 0.00000 0.03000 0.00000  100000 0.03000 0.00000
Bank Sta=0,100000
XS Rating Curve= 0 ,0
Exp/Cntr=0,0

Type RM Length L Ch R = 1 ,960     ,5,5,5
#Sta/Elev= 4
 0.00000 4.99055 0.00000-0.00945  100000-0.00945  100000 4.99055
#Mann= 3 ,0,0
 0.00000 0.03000 0.00000 0.00000 0.03000 0.00000  100000 0.03000 0.00000
Bank Sta=0,100000
XS Rating Curve= 0 ,0
Exp/Cntr=0,0

Type RM Length L Ch R = 1 ,955     ,5,5,5
#Sta/Elev= 4
 0.00000 4.98915 0.00000-0.01085  100000-0.01085  100000 4.98915
#Mann= 3 ,0,0
 0.00000 0.03000 0.00000 0.00000 0.03000 0.00000  100000 0.03000 0.00000
Bank Sta=0,100000
XS Rating Curve= 0 ,0
Exp/Cntr=0,0

Type RM Length L Ch R = 1 ,950     ,5,5,5
#Sta/Elev= 4
 0.00000 4.98768 0.00000-0.01232  100000-0.01232  100000 4.98768
#Mann= 3 ,0,0
 0.00000 0.03000 0.00000 0.00000 0.03000 0.00000  100000 0.03000 0.00000
Bank Sta=0,100000
XS Rating Curve= 0 ,0
Exp/Cntr=0,0

Type RM Length L Ch R = 1 ,945     ,5,5,5
#Sta/Elev= 4
 0.00000 4.98616 0.00000-0.01384  100000-0.01384  100000 4.98616
#Mann= 3 ,0,0
 0.00000 0.03000 0.00000 0.00000 0.03000 0.00000  100000 0.03000 0.00000
Bank Sta=0,100000
XS Rating Curve= 0 ,0
Exp/Cntr=0,0

Type RM Length L Ch R = 1 ,940     ,5,5,5
#Sta/Elev= 4
 0.00000 4.98457 0.00000-0.01543  100000-0.01543  100000 4.98457
#Mann= 3 ,0,0
 0.00000 0.03000 0.00000 0.00000 0.03000 0.00000  100000 0.03000 0.00000
Bank Sta=0,100000
XS Rating Curve= 0 ,0
Exp/Cntr=0,0

Type RM Length L Ch R = 1 ,935     ,5,5,5
#Sta/Elev= 4
 0.00000 4.98292 0.00000-0.01708  100000-0.01708  100000 4.98292
#Mann= 3 ,0,0
 0.00000 0.03000 0.00000 0.00000 0.03000 0.00000  100000 0.03000 0.00000
Bank Sta=0,100000
XS Rating Curve= 0 ,0
Exp/Cntr=0,0

Type RM Length L Ch R = 1 ,930     ,5,5,5
#Sta/Elev= 4
 0.00000  4.9812 0.00000-0.01880  100000-0.01880  100000  4.9812
#Mann= 3 ,0,0
 0.00000 0.03000 0.00000 0.00000 0.03000 0.00000  100000 0.03000 0.00000
Bank Sta=0,100000
XS Rating Curve= 0 ,0
Exp/Cntr=0,0

Type RM Length L Ch R = 1 ,925     ,5,5,5
#Sta/Elev= 4
 0.00000  4.9794 0.00000-0.02060  100000-0.02060  100000  4.9794
#Mann= 3 ,0,0
 0.00000 0.03000 0.00000 0.00000 0.03000 0.00000  100000 0.03000 0.00000
Bank Sta=0,100000
XS Rating Curve= 0 ,0
Exp/Cntr=0,0

Type RM Length L Ch R = 1 ,920     ,5,5,5
#Sta/Elev= 4
 0.00000 4.97753 0.00000-0.02247  100000-0.02247  100000 4.97753
#Mann= 3 ,0,0
 0.00000 0.03000 0.00000 0.00000 0.03000 0.00000  100000 0.03000 0.00000
Bank Sta=0,100000
XS Rating Curve= 0 ,0
Exp/Cntr=0,0

Type RM Length L Ch R = 1 ,915     ,5,5,5
#Sta/Elev= 4
 0.00000 4.97558 0.00000-0.02442  100000-0.02442  100000 4.97558
#Mann= 3 ,0,0
 0.00000 0.03000 0.00000 0.00000 0.03000 0.00000  100000 0.03000 0.00000
Bank Sta=0,100000
XS Rating Curve= 0 ,0
Exp/Cntr=0,0

Type RM Length L Ch R = 1 ,910     ,5,5,5
#Sta/Elev= 4
 0.00000 4.97355 0.00000-0.02645  100000-0.02645  100000 4.97355
#Mann= 3 ,0,0
 0.00000 0.03000 0.00000 0.00000 0.03000 0.00000  100000 0.03000 0.00000
Bank Sta=0,100000
XS Rating Curve= 0 ,0
Exp/Cntr=0,0

Type RM Length L Ch R = 1 ,905     ,5,5,5
#Sta/Elev= 4
 0.00000 4.97143 0.00000-0.02857  100000-0.02857  100000 4.97143
#Mann= 3 ,0,0
 0.00000 0.03000 0.00000 0.00000 0.03000 0.00000  100000 0.03000 0.00000
Bank Sta=0,100000
XS Rating Curve= 0 ,0
Exp/Cntr=0,0

Type RM Length L Ch R = 1 ,900     ,5,5,5
#Sta/Elev= 4
 0.00000 4.96923 0.00000-0.03077  100000-0.03077  100000 4.96923
#Mann= 3 ,0,0
 0.00000 0.03000 0.00000 0.00000 0.03000 0.00000  100000 0.03000 0.00000
Bank Sta=0,100000
XS Rating Curve= 0 ,0
Exp/Cntr=0,0

Type RM Length L Ch R = 1 ,895     ,5,5,5
#Sta/Elev= 4
 0.00000 4.96693 0.00000-0.03307  100000-0.03307  100000 4.96693
#Mann= 3 ,0,0
 0.00000 0.03000 0.00000 0.00000 0.03000 0.00000  100000 0.03000 0.00000
Bank Sta=0,100000
XS Rating Curve= 0 ,0
Exp/Cntr=0,0

Type RM Length L Ch R = 1 ,890     ,5,5,5
#Sta/Elev= 4
 0.00000 4.96455 0.00000-0.03545  100000-0.03545  100000 4.96455
#Mann= 3 ,0,0
 0.00000 0.03000 0.00000 0.00000 0.03000 0.00000  100000 0.03000 0.00000
Bank Sta=0,100000
XS Rating Curve= 0 ,0
Exp/Cntr=0,0

Type RM Length L Ch R = 1 ,885     ,5,5,5
#Sta/Elev= 4
 0.00000 4.96206 0.00000-0.03794  100000-0.03794  100000 4.96206
#Mann= 3 ,0,0
 0.00000 0.03000 0.00000 0.00000 0.03000 0.00000  100000 0.03000 0.00000
Bank Sta=0,100000
XS Rating Curve= 0 ,0
Exp/Cntr=0,0

Type RM Length L Ch R = 1 ,880     ,5,5,5
#Sta/Elev= 4
 0.00000 4.95948 0.00000-0.04052  100000-0.04052  100000 4.95948
#Mann= 3 ,0,0
 0.00000 0.03000 0.00000 0.00000 0.03000 0.00000  100000 0.03000 0.00000
Bank Sta=0,100000
XS Rating Curve= 0 ,0
Exp/Cntr=0,0

Type RM Length L Ch R = 1 ,875     ,5,5,5
#Sta/Elev= 4
 0.00000  4.9568 0.00000-0.04320  100000-0.04320  100000  4.9568
#Mann= 3 ,0,0
 0.00000 0.03000 0.00000 0.00000 0.03000 0.00000  100000 0.03000 0.00000
Bank Sta=0,100000
XS Rating Curve= 0 ,0
Exp/Cntr=0,0

Type RM Length L Ch R = 1 ,870     ,5,5,5
#Sta/Elev= 4
 0.00000 4.95401 0.00000-0.04599  100000-0.04599  100000 4.95401
#Mann= 3 ,0,0
 0.00000 0.03000 0.00000 0.00000 0.03000 0.00000  100000 0.03000 0.00000
Bank Sta=0,100000
XS Rating Curve= 0 ,0
Exp/Cntr=0,0

Type RM Length L Ch R = 1 ,865     ,5,5,5
#Sta/Elev= 4
 0.00000 4.95111 0.00000-0.04889  100000-0.04889  100000 4.95111
#Mann= 3 ,0,0
 0.00000 0.03000 0.00000 0.00000 0.03000 0.00000  100000 0.03000 0.00000
Bank Sta=0,100000
XS Rating Curve= 0 ,0
Exp/Cntr=0,0

Type RM Length L Ch R = 1 ,860     ,5,5,5
#Sta/Elev= 4
 0.00000 4.94811 0.00000-0.05189  100000-0.05189  100000 4.94811
#Mann= 3 ,0,0
 0.00000 0.03000 0.00000 0.00000 0.03000 0.00000  100000 0.03000 0.00000
Bank Sta=0,100000
XS Rating Curve= 0 ,0
Exp/Cntr=0,0

Type RM Length L Ch R = 1 ,855     ,5,5,5
#Sta/Elev= 4
 0.00000 4.94499 0.00000-0.05501  100000-0.05501  100000 4.94499
#Mann= 3 ,0,0
 0.00000 0.03000 0.00000 0.00000 0.03000 0.00000  100000 0.03000 0.00000
Bank Sta=0,100000
XS Rating Curve= 0 ,0
Exp/Cntr=0,0

Type RM Length L Ch R = 1 ,850     ,5,5,5
#Sta/Elev= 4
 0.00000 4.94176 0.00000-0.05824  100000-0.05824  100000 4.94176
#Mann= 3 ,0,0
 0.00000 0.03000 0.00000 0.00000 0.03000 0.00000  100000 0.03000 0.00000
Bank Sta=0,100000
XS Rating Curve= 0 ,0
Exp/Cntr=0,0

Type RM Length L Ch R = 1 ,845     ,5,5,5
#Sta/Elev= 4
 0.00000 4.93841 0.00000-0.06159  100000-0.06159  100000 4.93841
#Mann= 3 ,0,0
 0.00000 0.03000 0.00000 0.00000 0.03000 0.00000  100000 0.03000 0.00000
Bank Sta=0,100000
XS Rating Curve= 0 ,0
Exp/Cntr=0,0

Type RM Length L Ch R = 1 ,840     ,5,5,5
#Sta/Elev= 4
 0.00000 4.93495 0.00000-0.06505  100000-0.06505  100000 4.93495
#Mann= 3 ,0,0
 0.00000 0.03000 0.00000 0.00000 0.03000 0.00000  100000 0.03000 0.00000
Bank Sta=0,100000
XS Rating Curve= 0 ,0
Exp/Cntr=0,0

Type RM Length L Ch R = 1 ,835     ,5,5,5
#Sta/Elev= 4
 0.00000 4.93136 0.00000-0.06864  100000-0.06864  100000 4.93136
#Mann= 3 ,0,0
 0.00000 0.03000 0.00000 0.00000 0.03000 0.00000  100000 0.03000 0.00000
Bank Sta=0,100000
XS Rating Curve= 0 ,0
Exp/Cntr=0,0

Type RM Length L Ch R = 1 ,830     ,5,5,5
#Sta/Elev= 4
 0.00000 4.92765 0.00000-0.07235  100000-0.07235  100000 4.92765
#Mann= 3 ,0,0
 0.00000 0.03000 0.00000 0.00000 0.03000 0.00000  100000 0.03000 0.00000
Bank Sta=0,100000
XS Rating Curve= 0 ,0
Exp/Cntr=0,0

Type RM Length L Ch R = 1 ,825     ,5,5,5
#Sta/Elev= 4
 0.00000 4.92382 0.00000-0.07618  100000-0.07618  100000 4.92382
#Mann= 3 ,0,0
 0.00000 0.03000 0.00000 0.00000 0.03000 0.00000  100000 0.03000 0.00000
Bank Sta=0,100000
XS Rating Curve= 0 ,0
Exp/Cntr=0,0

Type RM Length L Ch R = 1 ,820     ,5,5,5
#Sta/Elev= 4
 0.00000 4.91986 0.00000-0.08014  100000-0.08014  100000 4.91986
#Mann= 3 ,0,0
 0.00000 0.03000 0.00000 0.00000 0.03000 0.00000  100000 0.03000 0.00000
Bank Sta=0,100000
XS Rating Curve= 0 ,0
Exp/Cntr=0,0

Type RM Length L Ch R = 1 ,815     ,5,5,5
#Sta/Elev= 4
 0.00000 4.91578 0.00000-0.08422  100000-0.08422  100000 4.91578
#Mann= 3 ,0,0
 0.00000 0.03000 0.00000 0.00000 0.03000 0.00000  100000 0.03000 0.00000
Bank Sta=0,100000
XS Rating Curve= 0 ,0
Exp/Cntr=0,0

Type RM Length L Ch R = 1 ,810     ,5,5,5
#Sta/Elev= 4
 0.00000 4.91158 0.00000-0.08842  100000-0.08842  100000 4.91158
#Mann= 3 ,0,0
 0.00000 0.03000 0.00000 0.00000 0.03000 0.00000  100000 0.03000 0.00000
Bank Sta=0,100000
XS Rating Curve= 0 ,0
Exp/Cntr=0,0

Type RM Length L Ch R = 1 ,805     ,5,5,5
#Sta/Elev= 4
 0.00000 4.90724 0.00000-0.09276  100000-0.09276  100000 4.90724
#Mann= 3 ,0,0
 0.00000 0.03000 0.00000 0.00000 0.03000 0.00000  100000 0.03000 0.00000
Bank Sta=0,100000
XS Rating Curve= 0 ,0
Exp/Cntr=0,0

Type RM Length L Ch R = 1 ,800     ,5,5,5
#Sta/Elev= 4
 0.00000 4.90278 0.00000-0.09722  100000-0.09722  100000 4.90278
#Mann= 3 ,0,0
 0.00000 0.03000 0.00000 0.00000 0.03000 0.00000  100000 0.03000 0.00000
Bank Sta=0,100000
XS Rating Curve= 0 ,0
Exp/Cntr=0,0

Type RM Length L Ch R = 1 ,795     ,5,5,5
#Sta/Elev= 4
 0.00000  4.8982 0.00000-0.10180  100000-0.10180  100000  4.8982
#Mann= 3 ,0,0
 0.00000 0.03000 0.00000 0.00000 0.03000 0.00000  100000 0.03000 0.00000
Bank Sta=0,100000
XS Rating Curve= 0 ,0
Exp/Cntr=0,0

Type RM Length L Ch R = 1 ,790     ,5,5,5
#Sta/Elev= 4
 0.00000 4.89349 0.00000-0.10651  100000-0.10651  100000 4.89349
#Mann= 3 ,0,0
 0.00000 0.03000 0.00000 0.00000 0.03000 0.00000  100000 0.03000 0.00000
Bank Sta=0,100000
XS Rating Curve= 0 ,0
Exp/Cntr=0,0

Type RM Length L Ch R = 1 ,785     ,5,5,5
#Sta/Elev= 4
 0.00000 4.88865 0.00000-0.11135  100000-0.11135  100000 4.88865
#Mann= 3 ,0,0
 0.00000 0.03000 0.00000 0.00000 0.03000 0.00000  100000 0.03000 0.00000
Bank Sta=0,100000
XS Rating Curve= 0 ,0
Exp/Cntr=0,0

Type RM Length L Ch R = 1 ,780     ,5,5,5
#Sta/Elev= 4
 0.00000 4.88369 0.00000-0.11631  100000-0.11631  100000 4.88369
#Mann= 3 ,0,0
 0.00000 0.03000 0.00000 0.00000 0.03000 0.00000  100000 0.03000 0.00000
Bank Sta=0,100000
XS Rating Curve= 0 ,0
Exp/Cntr=0,0

Type RM Length L Ch R = 1 ,775     ,5,5,5
#Sta/Elev= 4
 0.00000 4.87862 0.00000-0.12138  100000-0.12138  100000 4.87862
#Mann= 3 ,0,0
 0.00000 0.03000 0.00000 0.00000 0.03000 0.00000  100000 0.03000 0.00000
Bank Sta=0,100000
XS Rating Curve= 0 ,0
Exp/Cntr=0,0

Type RM Length L Ch R = 1 ,770     ,5,5,5
#Sta/Elev= 4
 0.00000 4.87342 0.00000-0.12658  100000-0.12658  100000 4.87342
#Mann= 3 ,0,0
 0.00000 0.03000 0.00000 0.00000 0.03000 0.00000  100000 0.03000 0.00000
Bank Sta=0,100000
XS Rating Curve= 0 ,0
Exp/Cntr=0,0

Type RM Length L Ch R = 1 ,765     ,5,5,5
#Sta/Elev= 4
 0.00000  4.8681 0.00000-0.13190  100000-0.13190  100000  4.8681
#Mann= 3 ,0,0
 0.00000 0.03000 0.00000 0.00000 0.03000 0.00000  100000 0.03000 0.00000
Bank Sta=0,100000
XS Rating Curve= 0 ,0
Exp/Cntr=0,0

Type RM Length L Ch R = 1 ,760     ,5,5,5
#Sta/Elev= 4
 0.00000 4.86267 0.00000-0.13733  100000-0.13733  100000 4.86267
#Mann= 3 ,0,0
 0.00000 0.03000 0.00000 0.00000 0.03000 0.00000  100000 0.03000 0.00000
Bank Sta=0,100000
XS Rating Curve= 0 ,0
Exp/Cntr=0,0

Type RM Length L Ch R = 1 ,755     ,5,5,5
#Sta/Elev= 4
 0.00000 4.85713 0.00000-0.14287  100000-0.14287  100000 4.85713
#Mann= 3 ,0,0
 0.00000 0.03000 0.00000 0.00000 0.03000 0.00000  100000 0.03000 0.00000
Bank Sta=0,100000
XS Rating Curve= 0 ,0
Exp/Cntr=0,0

Type RM Length L Ch R = 1 ,750     ,5,5,5
#Sta/Elev= 4
 0.00000 4.85148 0.00000-0.14852  100000-0.14852  100000 4.85148
#Mann= 3 ,0,0
 0.00000 0.03000 0.00000 0.00000 0.03000 0.00000  100000 0.03000 0.00000
Bank Sta=0,100000
XS Rating Curve= 0 ,0
Exp/Cntr=0,0

Type RM Length L Ch R = 1 ,745     ,5,5,5
#Sta/Elev= 4
 0.00000 4.84573 0.00000-0.15427  100000-0.15427  100000 4.84573
#Mann= 3 ,0,0
 0.00000 0.03000 0.00000 0.00000 0.03000 0.00000  100000 0.03000 0.00000
Bank Sta=0,100000
XS Rating Curve= 0 ,0
Exp/Cntr=0,0

Type RM Length L Ch R = 1 ,740     ,5,5,5
#Sta/Elev= 4
 0.00000 4.83988 0.00000-0.16012  100000-0.16012  100000 4.83988
#Mann= 3 ,0,0
 0.00000 0.03000 0.00000 0.00000 0.03000 0.00000  100000 0.03000 0.00000
Bank Sta=0,100000
XS Rating Curve= 0 ,0
Exp/Cntr=0,0

Type RM Length L Ch R = 1 ,735     ,5,5,5
#Sta/Elev= 4
 0.00000 4.83393 0.00000-0.16607  100000-0.16607  100000 4.83393
#Mann= 3 ,0,0
 0.00000 0.03000 0.00000 0.00000 0.03000 0.00000  100000 0.03000 0.00000
Bank Sta=0,100000
XS Rating Curve= 0 ,0
Exp/Cntr=0,0

Type RM Length L Ch R = 1 ,730     ,5,5,5
#Sta/Elev= 4
 0.00000  4.8279 0.00000-0.17210  100000-0.17210  100000  4.8279
#Mann= 3 ,0,0
 0.00000 0.03000 0.00000 0.00000 0.03000 0.00000  100000 0.03000 0.00000
Bank Sta=0,100000
XS Rating Curve= 0 ,0
Exp/Cntr=0,0

Type RM Length L Ch R = 1 ,725     ,5,5,5
#Sta/Elev= 4
 0.00000 4.82179 0.00000-0.17821  100000-0.17821  100000 4.82179
#Mann= 3 ,0,0
 0.00000 0.03000 0.00000 0.00000 0.03000 0.00000  100000 0.03000 0.00000
Bank Sta=0,100000
XS Rating Curve= 0 ,0
Exp/Cntr=0,0

Type RM Length L Ch R = 1 ,720     ,5,5,5
#Sta/Elev= 4
 0.00000 4.81559 0.00000-0.18441  100000-0.18441  100000 4.81559
#Mann= 3 ,0,0
 0.00000 0.03000 0.00000 0.00000 0.03000 0.00000  100000 0.03000 0.00000
Bank Sta=0,100000
XS Rating Curve= 0 ,0
Exp/Cntr=0,0

Type RM Length L Ch R = 1 ,715     ,5,5,5
#Sta/Elev= 4
 0.00000 4.80933 0.00000-0.19067  100000-0.19067  100000 4.80933
#Mann= 3 ,0,0
 0.00000 0.03000 0.00000 0.00000 0.03000 0.00000  100000 0.03000 0.00000
Bank Sta=0,100000
XS Rating Curve= 0 ,0
Exp/Cntr=0,0

Type RM Length L Ch R = 1 ,710     ,5,5,5
#Sta/Elev= 4
 0.00000 4.80301 0.00000-0.19699  100000-0.19699  100000 4.80301
#Mann= 3 ,0,0
 0.00000 0.03000 0.00000 0.00000 0.03000 0.00000  100000 0.03000 0.00000
Bank Sta=0,100000
XS Rating Curve= 0 ,0
Exp/Cntr=0,0

Type RM Length L Ch R = 1 ,705     ,5,5,5
#Sta/Elev= 4
 0.00000 4.79663 0.00000-0.20337  100000-0.20337  100000 4.79663
#Mann= 3 ,0,0
 0.00000 0.03000 0.00000 0.00000 0.03000 0.00000  100000 0.03000 0.00000
Bank Sta=0,100000
XS Rating Curve= 0 ,0
Exp/Cntr=0,0

Type RM Length L Ch R = 1 ,700     ,5,5,5
#Sta/Elev= 4
 0.00000  4.7902 0.00000-0.20980  100000-0.20980  100000  4.7902
#Mann= 3 ,0,0
 0.00000 0.03000 0.00000 0.00000 0.03000 0.00000  100000 0.03000 0.00000
Bank Sta=0,100000
XS Rating Curve= 0 ,0
Exp/Cntr=0,0

Type RM Length L Ch R = 1 ,695     ,5,5,5
#Sta/Elev= 4
 0.00000 4.78373 0.00000-0.21627  100000-0.21627  100000 4.78373
#Mann= 3 ,0,0
 0.00000 0.03000 0.00000 0.00000 0.03000 0.00000  100000 0.03000 0.00000
Bank Sta=0,100000
XS Rating Curve= 0 ,0
Exp/Cntr=0,0

Type RM Length L Ch R = 1 ,690     ,5,5,5
#Sta/Elev= 4
 0.00000 4.77723 0.00000-0.22277  100000-0.22277  100000 4.77723
#Mann= 3 ,0,0
 0.00000 0.03000 0.00000 0.00000 0.03000 0.00000  100000 0.03000 0.00000
Bank Sta=0,100000
XS Rating Curve= 0 ,0
Exp/Cntr=0,0

Type RM Length L Ch R = 1 ,685     ,5,5,5
#Sta/Elev= 4
 0.00000 4.77072 0.00000-0.22928  100000-0.22928  100000 4.77072
#Mann= 3 ,0,0
 0.00000 0.03000 0.00000 0.00000 0.03000 0.00000  100000 0.03000 0.00000
Bank Sta=0,100000
XS Rating Curve= 0 ,0
Exp/Cntr=0,0

Type RM Length L Ch R = 1 ,680     ,5,5,5
#Sta/Elev= 4
 0.00000 4.76418 0.00000-0.23582  100000-0.23582  100000 4.76418
#Mann= 3 ,0,0
 0.00000 0.03000 0.00000 0.00000 0.03000 0.00000  100000 0.03000 0.00000
Bank Sta=0,100000
XS Rating Curve= 0 ,0
Exp/Cntr=0,0

Type RM Length L Ch R = 1 ,675     ,5,5,5
#Sta/Elev= 4
 0.00000 4.75765 0.00000-0.24235  100000-0.24235  100000 4.75765
#Mann= 3 ,0,0
 0.00000 0.03000 0.00000 0.00000 0.03000 0.00000  100000 0.03000 0.00000
Bank Sta=0,100000
XS Rating Curve= 0 ,0
Exp/Cntr=0,0

Type RM Length L Ch R = 1 ,670     ,5,5,5
#Sta/Elev= 4
 0.00000 4.75112 0.00000-0.24888  100000-0.24888  100000 4.75112
#Mann= 3 ,0,0
 0.00000 0.03000 0.00000 0.00000 0.03000 0.00000  100000 0.03000 0.00000
Bank Sta=0,100000
XS Rating Curve= 0 ,0
Exp/Cntr=0,0

Type RM Length L Ch R = 1 ,665     ,5,5,5
#Sta/Elev= 4
 0.00000 4.74462 0.00000-0.25538  100000-0.25538  100000 4.74462
#Mann= 3 ,0,0
 0.00000 0.03000 0.00000 0.00000 0.03000 0.00000  100000 0.03000 0.00000
Bank Sta=0,100000
XS Rating Curve= 0 ,0
Exp/Cntr=0,0

Type RM Length L Ch R = 1 ,660     ,5,5,5
#Sta/Elev= 4
 0.00000 4.73814 0.00000-0.26186  100000-0.26186  100000 4.73814
#Mann= 3 ,0,0
 0.00000 0.03000 0.00000 0.00000 0.03000 0.00000  100000 0.03000 0.00000
Bank Sta=0,100000
XS Rating Curve= 0 ,0
Exp/Cntr=0,0

Type RM Length L Ch R = 1 ,655     ,5,5,5
#Sta/Elev= 4
 0.00000 4.73169 0.00000-0.26831  100000-0.26831  100000 4.73169
#Mann= 3 ,0,0
 0.00000 0.03000 0.00000 0.00000 0.03000 0.00000  100000 0.03000 0.00000
Bank Sta=0,100000
XS Rating Curve= 0 ,0
Exp/Cntr=0,0

Type RM Length L Ch R = 1 ,650     ,5,5,5
#Sta/Elev= 4
 0.00000  4.7253 0.00000-0.27470  100000-0.27470  100000  4.7253
#Mann= 3 ,0,0
 0.00000 0.03000 0.00000 0.00000 0.03000 0.00000  100000 0.03000 0.00000
Bank Sta=0,100000
XS Rating Curve= 0 ,0
Exp/Cntr=0,0

Type RM Length L Ch R = 1 ,645     ,5,5,5
#Sta/Elev= 4
 0.00000 4.71897 0.00000-0.28103  100000-0.28103  100000 4.71897
#Mann= 3 ,0,0
 0.00000 0.03000 0.00000 0.00000 0.03000 0.00000  100000 0.03000 0.00000
Bank Sta=0,100000
XS Rating Curve= 0 ,0
Exp/Cntr=0,0

Type RM Length L Ch R = 1 ,640     ,5,5,5
#Sta/Elev= 4
 0.00000 4.71271 0.00000-0.28729  100000-0.28729  100000 4.71271
#Mann= 3 ,0,0
 0.00000 0.03000 0.00000 0.00000 0.03000 0.00000  100000 0.03000 0.00000
Bank Sta=0,100000
XS Rating Curve= 0 ,0
Exp/Cntr=0,0

Type RM Length L Ch R = 1 ,635     ,5,5,5
#Sta/Elev= 4
 0.00000 4.70654 0.00000-0.29346  100000-0.29346  100000 4.70654
#Mann= 3 ,0,0
 0.00000 0.03000 0.00000 0.00000 0.03000 0.00000  100000 0.03000 0.00000
Bank Sta=0,100000
XS Rating Curve= 0 ,0
Exp/Cntr=0,0

Type RM Length L Ch R = 1 ,630     ,5,5,5
#Sta/Elev= 4
 0.00000 4.70046 0.00000-0.29954  100000-0.29954  100000 4.70046
#Mann= 3 ,0,0
 0.00000 0.03000 0.00000 0.00000 0.03000 0.00000  100000 0.03000 0.00000
Bank Sta=0,100000
XS Rating Curve= 0 ,0
Exp/Cntr=0,0

Type RM Length L Ch R = 1 ,625     ,5,5,5
#Sta/Elev= 4
 0.00000 4.69449 0.00000-0.30551  100000-0.30551  100000 4.69449
#Mann= 3 ,0,0
 0.00000 0.03000 0.00000 0.00000 0.03000 0.00000  100000 0.03000 0.00000
Bank Sta=0,100000
XS Rating Curve= 0 ,0
Exp/Cntr=0,0

Type RM Length L Ch R = 1 ,620     ,5,5,5
#Sta/Elev= 4
 0.00000 4.68863 0.00000-0.31137  100000-0.31137  100000 4.68863
#Mann= 3 ,0,0
 0.00000 0.03000 0.00000 0.00000 0.03000 0.00000  100000 0.03000 0.00000
Bank Sta=0,100000
XS Rating Curve= 0 ,0
Exp/Cntr=0,0

Type RM Length L Ch R = 1 ,615     ,5,5,5
#Sta/Elev= 4
 0.00000  4.6829 0.00000-0.31710  100000-0.31710  100000  4.6829
#Mann= 3 ,0,0
 0.00000 0.03000 0.00000 0.00000 0.03000 0.00000  100000 0.03000 0.00000
Bank Sta=0,100000
XS Rating Curve= 0 ,0
Exp/Cntr=0,0

Type RM Length L Ch R = 1 ,610     ,5,5,5
#Sta/Elev= 4
 0.00000 4.67732 0.00000-0.32268  100000-0.32268  100000 4.67732
#Mann= 3 ,0,0
 0.00000 0.03000 0.00000 0.00000 0.03000 0.00000  100000 0.03000 0.00000
Bank Sta=0,100000
XS Rating Curve= 0 ,0
Exp/Cntr=0,0

Type RM Length L Ch R = 1 ,605     ,5,5,5
#Sta/Elev= 4
 0.00000 4.67188 0.00000-0.32812  100000-0.32812  100000 4.67188
#Mann= 3 ,0,0
 0.00000 0.03000 0.00000 0.00000 0.03000 0.00000  100000 0.03000 0.00000
Bank Sta=0,100000
XS Rating Curve= 0 ,0
Exp/Cntr=0,0

Type RM Length L Ch R = 1 ,600     ,5,5,5
#Sta/Elev= 4
 0.00000 4.66661 0.00000-0.33339  100000-0.33339  100000 4.66661
#Mann= 3 ,0,0
 0.00000 0.03000 0.00000 0.00000 0.03000 0.00000  100000 0.03000 0.00000
Bank Sta=0,100000
XS Rating Curve= 0 ,0
Exp/Cntr=0,0

Type RM Length L Ch R = 1 ,595     ,5,5,5
#Sta/Elev= 4
 0.00000 4.66151 0.00000-0.33849  100000-0.33849  100000 4.66151
#Mann= 3 ,0,0
 0.00000 0.03000 0.00000 0.00000 0.03000 0.00000  100000 0.03000 0.00000
Bank Sta=0,100000
XS Rating Curve= 0 ,0
Exp/Cntr=0,0

Type RM Length L Ch R = 1 ,590     ,5,5,5
#Sta/Elev= 4
 0.00000  4.6566 0.00000-0.34340  100000-0.34340  100000  4.6566
#Mann= 3 ,0,0
 0.00000 0.03000 0.00000 0.00000 0.03000 0.00000  100000 0.03000 0.00000
Bank Sta=0,100000
XS Rating Curve= 0 ,0
Exp/Cntr=0,0

Type RM Length L Ch R = 1 ,585     ,5,5,5
#Sta/Elev= 4
 0.00000 4.65188 0.00000-0.34812  100000-0.34812  100000 4.65188
#Mann= 3 ,0,0
 0.00000 0.03000 0.00000 0.00000 0.03000 0.00000  100000 0.03000 0.00000
Bank Sta=0,100000
XS Rating Curve= 0 ,0
Exp/Cntr=0,0

Type RM Length L Ch R = 1 ,580     ,5,5,5
#Sta/Elev= 4
 0.00000 4.64736 0.00000-0.35264  100000-0.35264  100000 4.64736
#Mann= 3 ,0,0
 0.00000 0.03000 0.00000 0.00000 0.03000 0.00000  100000 0.03000 0.00000
Bank Sta=0,100000
XS Rating Curve= 0 ,0
Exp/Cntr=0,0

Type RM Length L Ch R = 1 ,575     ,5,5,5
#Sta/Elev= 4
 0.00000 4.64306 0.00000-0.35694  100000-0.35694  100000 4.64306
#Mann= 3 ,0,0
 0.00000 0.03000 0.00000 0.00000 0.03000 0.00000  100000 0.03000 0.00000
Bank Sta=0,100000
XS Rating Curve= 0 ,0
Exp/Cntr=0,0

Type RM Length L Ch R = 1 ,570     ,5,5,5
#Sta/Elev= 4
 0.00000 4.63898 0.00000-0.36102  100000-0.36102  100000 4.63898
#Mann= 3 ,0,0
 0.00000 0.03000 0.00000 0.00000 0.03000 0.00000  100000 0.03000 0.00000
Bank Sta=0,100000
XS Rating Curve= 0 ,0
Exp/Cntr=0,0

Type RM Length L Ch R = 1 ,565     ,5,5,5
#Sta/Elev= 4
 0.00000 4.63513 0.00000-0.36487  100000-0.36487  100000 4.63513
#Mann= 3 ,0,0
 0.00000 0.03000 0.00000 0.00000 0.03000 0.00000  100000 0.03000 0.00000
Bank Sta=0,100000
XS Rating Curve= 0 ,0
Exp/Cntr=0,0

Type RM Length L Ch R = 1 ,560     ,5,5,5
#Sta/Elev= 4
 0.00000 4.63153 0.00000-0.36847  100000-0.36847  100000 4.63153
#Mann= 3 ,0,0
 0.00000 0.03000 0.00000 0.00000 0.03000 0.00000  100000 0.03000 0.00000
Bank Sta=0,100000
XS Rating Curve= 0 ,0
Exp/Cntr=0,0

Type RM Length L Ch R = 1 ,555     ,5,5,5
#Sta/Elev= 4
 0.00000 4.62817 0.00000-0.37183  100000-0.37183  100000 4.62817
#Mann= 3 ,0,0
 0.00000 0.03000 0.00000 0.00000 0.03000 0.00000  100000 0.03000 0.00000
Bank Sta=0,100000
XS Rating Curve= 0 ,0
Exp/Cntr=0,0

Type RM Length L Ch R = 1 ,550     ,5,5,5
#Sta/Elev= 4
 0.00000 4.62506 0.00000-0.37494  100000-0.37494  100000 4.62506
#Mann= 3 ,0,0
 0.00000 0.03000 0.00000 0.00000 0.03000 0.00000  100000 0.03000 0.00000
Bank Sta=0,100000
XS Rating Curve= 0 ,0
Exp/Cntr=0,0

Type RM Length L Ch R = 1 ,545     ,5,5,5
#Sta/Elev= 4
 0.00000 4.62222 0.00000-0.37778  100000-0.37778  100000 4.62222
#Mann= 3 ,0,0
 0.00000 0.03000 0.00000 0.00000 0.03000 0.00000  100000 0.03000 0.00000
Bank Sta=0,100000
XS Rating Curve= 0 ,0
Exp/Cntr=0,0

Type RM Length L Ch R = 1 ,540     ,5,5,5
#Sta/Elev= 4
 0.00000 4.61965 0.00000-0.38035  100000-0.38035  100000 4.61965
#Mann= 3 ,0,0
 0.00000 0.03000 0.00000 0.00000 0.03000 0.00000  100000 0.03000 0.00000
Bank Sta=0,100000
XS Rating Curve= 0 ,0
Exp/Cntr=0,0

Type RM Length L Ch R = 1 ,535     ,5,5,5
#Sta/Elev= 4
 0.00000 4.61735 0.00000-0.38265  100000-0.38265  100000 4.61735
#Mann= 3 ,0,0
 0.00000 0.03000 0.00000 0.00000 0.03000 0.00000  100000 0.03000 0.00000
Bank Sta=0,100000
XS Rating Curve= 0 ,0
Exp/Cntr=0,0

Type RM Length L Ch R = 1 ,530     ,5,5,5
#Sta/Elev= 4
 0.00000 4.61534 0.00000-0.38466  100000-0.38466  100000 4.61534
#Mann= 3 ,0,0
 0.00000 0.03000 0.00000 0.00000 0.03000 0.00000  100000 0.03000 0.00000
Bank Sta=0,100000
XS Rating Curve= 0 ,0
Exp/Cntr=0,0

Type RM Length L Ch R = 1 ,525     ,5,5,5
#Sta/Elev= 4
 0.00000  4.6136 0.00000-0.38640  100000-0.38640  100000  4.6136
#Mann= 3 ,0,0
 0.00000 0.03000 0.00000 0.00000 0.03000 0.00000  100000 0.03000 0.00000
Bank Sta=0,100000
XS Rating Curve= 0 ,0
Exp/Cntr=0,0

Type RM Length L Ch R = 1 ,520     ,5,5,5
#Sta/Elev= 4
 0.00000 4.61215 0.00000-0.38785  100000-0.38785  100000 4.61215
#Mann= 3 ,0,0
 0.00000 0.03000 0.00000 0.00000 0.03000 0.00000  100000 0.03000 0.00000
Bank Sta=0,100000
XS Rating Curve= 0 ,0
Exp/Cntr=0,0

Type RM Length L Ch R = 1 ,515     ,5,5,5
#Sta/Elev= 4
 0.00000   4.611 0.00000-0.38900  100000-0.38900  100000   4.611
#Mann= 3 ,0,0
 0.00000 0.03000 0.00000 0.00000 0.03000 0.00000  100000 0.03000 0.00000
Bank Sta=0,100000
XS Rating Curve= 0 ,0
Exp/Cntr=0,0

Type RM Length L Ch R = 1 ,510     ,5,5,5
#Sta/Elev= 4
 0.00000 4.61013 0.00000-0.38987  100000-0.38987  100000 4.61013
#Mann= 3 ,0,0
 0.00000 0.03000 0.00000 0.00000 0.03000 0.00000  100000 0.03000 0.00000
Bank Sta=0,100000
XS Rating Curve= 0 ,0
Exp/Cntr=0,0

Type RM Length L Ch R = 1 ,505     ,5,5,5
#Sta/Elev= 4
 0.00000 4.60956 0.00000-0.39044  100000-0.39044  100000 4.60956
#Mann= 3 ,0,0
 0.00000 0.03000 0.00000 0.00000 0.03000 0.00000  100000 0.03000 0.00000
Bank Sta=0,100000
XS Rating Curve= 0 ,0
Exp/Cntr=0,0

Type RM Length L Ch R = 1 ,500     ,5,5,5
#Sta/Elev= 4
 0.00000 4.60929 0.00000-0.39071  100000-0.39071  100000 4.60929
#Mann= 3 ,0,0
 0.00000 0.03000 0.00000 0.00000 0.03000 0.00000  100000 0.03000 0.00000
Bank Sta=0,100000
XS Rating Curve= 0 ,0
Exp/Cntr=0,0

Type RM Length L Ch R = 1 ,495     ,5,5,5
#Sta/Elev= 4
 0.00000 4.60931 0.00000-0.39069  100000-0.39069  100000 4.60931
#Mann= 3 ,0,0
 0.00000 0.03000 0.00000 0.00000 0.03000 0.00000  100000 0.03000 0.00000
Bank Sta=0,100000
XS Rating Curve= 0 ,0
Exp/Cntr=0,0

Type RM Length L Ch R = 1 ,490     ,5,5,5
#Sta/Elev= 4
 0.00000 4.60963 0.00000-0.39037  100000-0.39037  100000 4.60963
#Mann= 3 ,0,0
 0.00000 0.03000 0.00000 0.00000 0.03000 0.00000  100000 0.03000 0.00000
Bank Sta=0,100000
XS Rating Curve= 0 ,0
Exp/Cntr=0,0

Type RM Length L Ch R = 1 ,485     ,5,5,5
#Sta/Elev= 4
 0.00000 4.61024 0.00000-0.38976  100000-0.38976  100000 4.61024
#Mann= 3 ,0,0
 0.00000 0.03000 0.00000 0.00000 0.03000 0.00000  100000 0.03000 0.00000
Bank Sta=0,100000
XS Rating Curve= 0 ,0
Exp/Cntr=0,0

Type RM Length L Ch R = 1 ,480     ,5,5,5
#Sta/Elev= 4
 0.00000 4.61114 0.00000-0.38886  100000-0.38886  100000 4.61114
#Mann= 3 ,0,0
 0.00000 0.03000 0.00000 0.00000 0.03000 0.00000  100000 0.03000 0.00000
Bank Sta=0,100000
XS Rating Curve= 0 ,0
Exp/Cntr=0,0

Type RM Length L Ch R = 1 ,475     ,5,5,5
#Sta/Elev= 4
 0.00000 4.61233 0.00000-0.38767  100000-0.38767  100000 4.61233
#Mann= 3 ,0,0
 0.00000 0.03000 0.00000 0.00000 0.03000 0.00000  100000 0.03000 0.00000
Bank Sta=0,100000
XS Rating Curve= 0 ,0
Exp/Cntr=0,0

Type RM Length L Ch R = 1 ,470     ,5,5,5
#Sta/Elev= 4
 0.00000 4.61381 0.00000-0.38619  100000-0.38619  100000 4.61381
#Mann= 3 ,0,0
 0.00000 0.03000 0.00000 0.00000 0.03000 0.00000  100000 0.03000 0.00000
Bank Sta=0,100000
XS Rating Curve= 0 ,0
Exp/Cntr=0,0

Type RM Length L Ch R = 1 ,465     ,5,5,5
#Sta/Elev= 4
 0.00000 4.61557 0.00000-0.38443  100000-0.38443  100000 4.61557
#Mann= 3 ,0,0
 0.00000 0.03000 0.00000 0.00000 0.03000 0.00000  100000 0.03000 0.00000
Bank Sta=0,100000
XS Rating Curve= 0 ,0
Exp/Cntr=0,0

Type RM Length L Ch R = 1 ,460     ,5,5,5
#Sta/Elev= 4
 0.00000 4.61761 0.00000-0.38239  100000-0.38239  100000 4.61761
#Mann= 3 ,0,0
 0.00000 0.03000 0.00000 0.00000 0.03000 0.00000  100000 0.03000 0.00000
Bank Sta=0,100000
XS Rating Curve= 0 ,0
Exp/Cntr=0,0

Type RM Length L Ch R = 1 ,455     ,5,5,5
#Sta/Elev= 4
 0.00000 4.61992 0.00000-0.38008  100000-0.38008  100000 4.61992
#Mann= 3 ,0,0
 0.00000 0.03000 0.00000 0.00000 0.03000 0.00000  100000 0.03000 0.00000
Bank Sta=0,100000
XS Rating Curve= 0 ,0
Exp/Cntr=0,0

Type RM Length L Ch R = 1 ,450     ,5,5,5
#Sta/Elev= 4
 0.00000  4.6225 0.00000-0.37750  100000-0.37750  100000  4.6225
#Mann= 3 ,0,0
 0.00000 0.03000 0.00000 0.00000 0.03000 0.00000  100000 0.03000 0.00000
Bank Sta=0,100000
XS Rating Curve= 0 ,0
Exp/Cntr=0,0

Type RM Length L Ch R = 1 ,445     ,5,5,5
#Sta/Elev= 4
 0.00000 4.62534 0.00000-0.37466  100000-0.37466  100000 4.62534
#Mann= 3 ,0,0
 0.00000 0.03000 0.00000 0.00000 0.03000 0.00000  100000 0.03000 0.00000
Bank Sta=0,100000
XS Rating Curve= 0 ,0
Exp/Cntr=0,0

Type RM Length L Ch R = 1 ,440     ,5,5,5
#Sta/Elev= 4
 0.00000 4.62843 0.00000-0.37157  100000-0.37157  100000 4.62843
#Mann= 3 ,0,0
 0.00000 0.03000 0.00000 0.00000 0.03000 0.00000  100000 0.03000 0.00000
Bank Sta=0,100000
XS Rating Curve= 0 ,0
Exp/Cntr=0,0

Type RM Length L Ch R = 1 ,435     ,5,5,5
#Sta/Elev= 4
 0.00000 4.63177 0.00000-0.36823  100000-0.36823  100000 4.63177
#Mann= 3 ,0,0
 0.00000 0.03000 0.00000 0.00000 0.03000 0.00000  100000 0.03000 0.00000
Bank Sta=0,100000
XS Rating Curve= 0 ,0
Exp/Cntr=0,0

Type RM Length L Ch R = 1 ,430     ,5,5,5
#Sta/Elev= 4
 0.00000 4.63534 0.00000-0.36466  100000-0.36466  100000 4.63534
#Mann= 3 ,0,0
 0.00000 0.03000 0.00000 0.00000 0.03000 0.00000  100000 0.03000 0.00000
Bank Sta=0,100000
XS Rating Curve= 0 ,0
Exp/Cntr=0,0

Type RM Length L Ch R = 1 ,425     ,5,5,5
#Sta/Elev= 4
 0.00000 4.63914 0.00000-0.36086  100000-0.36086  100000 4.63914
#Mann= 3 ,0,0
 0.00000 0.03000 0.00000 0.00000 0.03000 0.00000  100000 0.03000 0.00000
Bank Sta=0,100000
XS Rating Curve= 0 ,0
Exp/Cntr=0,0

Type RM Length L Ch R = 1 ,420     ,5,5,5
#Sta/Elev= 4
 0.00000 4.64317 0.00000-0.35683  100000-0.35683  100000 4.64317
#Mann= 3 ,0,0
 0.00000 0.03000 0.00000 0.00000 0.03000 0.00000  100000 0.03000 0.00000
Bank Sta=0,100000
XS Rating Curve= 0 ,0
Exp/Cntr=0,0

Type RM Length L Ch R = 1 ,415     ,5,5,5
#Sta/Elev= 4
 0.00000  4.6474 0.00000-0.35260  100000-0.35260  100000  4.6474
#Mann= 3 ,0,0
 0.00000 0.03000 0.00000 0.00000 0.03000 0.00000  100000 0.03000 0.00000
Bank Sta=0,100000
XS Rating Curve= 0 ,0
Exp/Cntr=0,0

Type RM Length L Ch R = 1 ,410     ,5,5,5
#Sta/Elev= 4
 0.00000 4.65183 0.00000-0.34817  100000-0.34817  100000 4.65183
#Mann= 3 ,0,0
 0.00000 0.03000 0.00000 0.00000 0.03000 0.00000  100000 0.03000 0.00000
Bank Sta=0,100000
XS Rating Curve= 0 ,0
Exp/Cntr=0,0

Type RM Length L Ch R = 1 ,405     ,5,5,5
#Sta/Elev= 4
 0.00000 4.65645 0.00000-0.34355  100000-0.34355  100000 4.65645
#Mann= 3 ,0,0
 0.00000 0.03000 0.00000 0.00000 0.03000 0.00000  100000 0.03000 0.00000
Bank Sta=0,100000
XS Rating Curve= 0 ,0
Exp/Cntr=0,0

Type RM Length L Ch R = 1 ,400     ,5,5,5
#Sta/Elev= 4
 0.00000 4.66126 0.00000-0.33874  100000-0.33874  100000 4.66126
#Mann= 3 ,0,0
 0.00000 0.03000 0.00000 0.00000 0.03000 0.00000  100000 0.03000 0.00000
Bank Sta=0,100000
XS Rating Curve= 0 ,0
Exp/Cntr=0,0

Type RM Length L Ch R = 1 ,395     ,5,5,5
#Sta/Elev= 4
 0.00000 4.66623 0.00000-0.33377  100000-0.33377  100000 4.66623
#Mann= 3 ,0,0
 0.00000 0.03000 0.00000 0.00000 0.03000 0.00000  100000 0.03000 0.00000
Bank Sta=0,100000
XS Rating Curve= 0 ,0
Exp/Cntr=0,0

Type RM Length L Ch R = 1 ,390     ,5,5,5
#Sta/Elev= 4
 0.00000 4.67136 0.00000-0.32864  100000-0.32864  100000 4.67136
#Mann= 3 ,0,0
 0.00000 0.03000 0.00000 0.00000 0.03000 0.00000  100000 0.03000 0.00000
Bank Sta=0,100000
XS Rating Curve= 0 ,0
Exp/Cntr=0,0

Type RM Length L Ch R = 1 ,385     ,5,5,5
#Sta/Elev= 4
 0.00000 4.67663 0.00000-0.32337  100000-0.32337  100000 4.67663
#Mann= 3 ,0,0
 0.00000 0.03000 0.00000 0.00000 0.03000 0.00000  100000 0.03000 0.00000
Bank Sta=0,100000
XS Rating Curve= 0 ,0
Exp/Cntr=0,0

Type RM Length L Ch R = 1 ,380     ,5,5,5
#Sta/Elev= 4
 0.00000 4.68204 0.00000-0.31796  100000-0.31796  100000 4.68204
#Mann= 3 ,0,0
 0.00000 0.03000 0.00000 0.00000 0.03000 0.00000  100000 0.03000 0.00000
Bank Sta=0,100000
XS Rating Curve= 0 ,0
Exp/Cntr=0,0

Type RM Length L Ch R = 1 ,375     ,5,5,5
#Sta/Elev= 4
 0.00000 4.68757 0.00000-0.31243  100000-0.31243  100000 4.68757
#Mann= 3 ,0,0
 0.00000 0.03000 0.00000 0.00000 0.03000 0.00000  100000 0.03000 0.00000
Bank Sta=0,100000
XS Rating Curve= 0 ,0
Exp/Cntr=0,0

Type RM Length L Ch R = 1 ,370     ,5,5,5
#Sta/Elev= 4
 0.00000 4.69322 0.00000-0.30678  100000-0.30678  100000 4.69322
#Mann= 3 ,0,0
 0.00000 0.03000 0.00000 0.00000 0.03000 0.00000  100000 0.03000 0.00000
Bank Sta=0,100000
XS Rating Curve= 0 ,0
Exp/Cntr=0,0

Type RM Length L Ch R = 1 ,365     ,5,5,5
#Sta/Elev= 4
 0.00000 4.69896 0.00000-0.30104  100000-0.30104  100000 4.69896
#Mann= 3 ,0,0
 0.00000 0.03000 0.00000 0.00000 0.03000 0.00000  100000 0.03000 0.00000
Bank Sta=0,100000
XS Rating Curve= 0 ,0
Exp/Cntr=0,0

Type RM Length L Ch R = 1 ,360     ,5,5,5
#Sta/Elev= 4
 0.00000 4.70479 0.00000-0.29521  100000-0.29521  100000 4.70479
#Mann= 3 ,0,0
 0.00000 0.03000 0.00000 0.00000 0.03000 0.00000  100000 0.03000 0.00000
Bank Sta=0,100000
XS Rating Curve= 0 ,0
Exp/Cntr=0,0

Type RM Length L Ch R = 1 ,355     ,5,5,5
#Sta/Elev= 4
 0.00000  4.7107 0.00000-0.28930  100000-0.28930  100000  4.7107
#Mann= 3 ,0,0
 0.00000 0.03000 0.00000 0.00000 0.03000 0.00000  100000 0.03000 0.00000
Bank Sta=0,100000
XS Rating Curve= 0 ,0
Exp/Cntr=0,0

Type RM Length L Ch R = 1 ,350     ,5,5,5
#Sta/Elev= 4
 0.00000 4.71668 0.00000-0.28332  100000-0.28332  100000 4.71668
#Mann= 3 ,0,0
 0.00000 0.03000 0.00000 0.00000 0.03000 0.00000  100000 0.03000 0.00000
Bank Sta=0,100000
XS Rating Curve= 0 ,0
Exp/Cntr=0,0

Type RM Length L Ch R = 1 ,345     ,5,5,5
#Sta/Elev= 4
 0.00000 4.72271 0.00000-0.27729  100000-0.27729  100000 4.72271
#Mann= 3 ,0,0
 0.00000 0.03000 0.00000 0.00000 0.03000 0.00000  100000 0.03000 0.00000
Bank Sta=0,100000
XS Rating Curve= 0 ,0
Exp/Cntr=0,0

Type RM Length L Ch R = 1 ,340     ,5,5,5
#Sta/Elev= 4
 0.00000 4.72878 0.00000-0.27122  100000-0.27122  100000 4.72878
#Mann= 3 ,0,0
 0.00000 0.03000 0.00000 0.00000 0.03000 0.00000  100000 0.03000 0.00000
Bank Sta=0,100000
XS Rating Curve= 0 ,0
Exp/Cntr=0,0

Type RM Length L Ch R = 1 ,335     ,5,5,5
#Sta/Elev= 4
 0.00000 4.73488 0.00000-0.26512  100000-0.26512  100000 4.73488
#Mann= 3 ,0,0
 0.00000 0.03000 0.00000 0.00000 0.03000 0.00000  100000 0.03000 0.00000
Bank Sta=0,100000
XS Rating Curve= 0 ,0
Exp/Cntr=0,0

Type RM Length L Ch R = 1 ,330     ,5,5,5
#Sta/Elev= 4
 0.00000   4.741 0.00000-0.25900  100000-0.25900  100000   4.741
#Mann= 3 ,0,0
 0.00000 0.03000 0.00000 0.00000 0.03000 0.00000  100000 0.03000 0.00000
Bank Sta=0,100000
XS Rating Curve= 0 ,0
Exp/Cntr=0,0

Type RM Length L Ch R = 1 ,325     ,5,5,5
#Sta/Elev= 4
 0.00000 4.74713 0.00000-0.25287  100000-0.25287  100000 4.74713
#Mann= 3 ,0,0
 0.00000 0.03000 0.00000 0.00000 0.03000 0.00000  100000 0.03000 0.00000
Bank Sta=0,100000
XS Rating Curve= 0 ,0
Exp/Cntr=0,0

Type RM Length L Ch R = 1 ,320     ,5,5,5
#Sta/Elev= 4
 0.00000 4.75326 0.00000-0.24674  100000-0.24674  100000 4.75326
#Mann= 3 ,0,0
 0.00000 0.03000 0.00000 0.00000 0.03000 0.00000  100000 0.03000 0.00000
Bank Sta=0,100000
XS Rating Curve= 0 ,0
Exp/Cntr=0,0

Type RM Length L Ch R = 1 ,315     ,5,5,5
#Sta/Elev= 4
 0.00000 4.75937 0.00000-0.24063  100000-0.24063  100000 4.75937
#Mann= 3 ,0,0
 0.00000 0.03000 0.00000 0.00000 0.03000 0.00000  100000 0.03000 0.00000
Bank Sta=0,100000
XS Rating Curve= 0 ,0
Exp/Cntr=0,0

Type RM Length L Ch R = 1 ,310     ,5,5,5
#Sta/Elev= 4
 0.00000 4.76547 0.00000-0.23453  100000-0.23453  100000 4.76547
#Mann= 3 ,0,0
 0.00000 0.03000 0.00000 0.00000 0.03000 0.00000  100000 0.03000 0.00000
Bank Sta=0,100000
XS Rating Curve= 0 ,0
Exp/Cntr=0,0

Type RM Length L Ch R = 1 ,305     ,5,5,5
#Sta/Elev= 4
 0.00000 4.77154 0.00000-0.22846  100000-0.22846  100000 4.77154
#Mann= 3 ,0,0
 0.00000 0.03000 0.00000 0.00000 0.03000 0.00000  100000 0.03000 0.00000
Bank Sta=0,100000
XS Rating Curve= 0 ,0
Exp/Cntr=0,0

Type RM Length L Ch R = 1 ,300     ,5,5,5
#Sta/Elev= 4
 0.00000 4.77756 0.00000-0.22244  100000-0.22244  100000 4.77756
#Mann= 3 ,0,0
 0.00000 0.03000 0.00000 0.00000 0.03000 0.00000  100000 0.03000 0.00000
Bank Sta=0,100000
XS Rating Curve= 0 ,0
Exp/Cntr=0,0

Type RM Length L Ch R = 1 ,295     ,5,5,5
#Sta/Elev= 4
 0.00000 4.78354 0.00000-0.21646  100000-0.21646  100000 4.78354
#Mann= 3 ,0,0
 0.00000 0.03000 0.00000 0.00000 0.03000 0.00000  100000 0.03000 0.00000
Bank Sta=0,100000
XS Rating Curve= 0 ,0
Exp/Cntr=0,0

Type RM Length L Ch R = 1 ,290     ,5,5,5
#Sta/Elev= 4
 0.00000 4.78945 0.00000-0.21055  100000-0.21055  100000 4.78945
#Mann= 3 ,0,0
 0.00000 0.03000 0.00000 0.00000 0.03000 0.00000  100000 0.03000 0.00000
Bank Sta=0,100000
XS Rating Curve= 0 ,0
Exp/Cntr=0,0

Type RM Length L Ch R = 1 ,285     ,5,5,5
#Sta/Elev= 4
 0.00000 4.79531 0.00000-0.20469  100000-0.20469  100000 4.79531
#Mann= 3 ,0,0
 0.00000 0.03000 0.00000 0.00000 0.03000 0.00000  100000 0.03000 0.00000
Bank Sta=0,100000
XS Rating Curve= 0 ,0
Exp/Cntr=0,0

Type RM Length L Ch R = 1 ,280     ,5,5,5
#Sta/Elev= 4
 0.00000 4.80108 0.00000-0.19892  100000-0.19892  100000 4.80108
#Mann= 3 ,0,0
 0.00000 0.03000 0.00000 0.00000 0.03000 0.00000  100000 0.03000 0.00000
Bank Sta=0,100000
XS Rating Curve= 0 ,0
Exp/Cntr=0,0

Type RM Length L Ch R = 1 ,275     ,5,5,5
#Sta/Elev= 4
 0.00000 4.80678 0.00000-0.19322  100000-0.19322  100000 4.80678
#Mann= 3 ,0,0
 0.00000 0.03000 0.00000 0.00000 0.03000 0.00000  100000 0.03000 0.00000
Bank Sta=0,100000
XS Rating Curve= 0 ,0
Exp/Cntr=0,0

Type RM Length L Ch R = 1 ,270     ,5,5,5
#Sta/Elev= 4
 0.00000 4.81239 0.00000-0.18761  100000-0.18761  100000 4.81239
#Mann= 3 ,0,0
 0.00000 0.03000 0.00000 0.00000 0.03000 0.00000  100000 0.03000 0.00000
Bank Sta=0,100000
XS Rating Curve= 0 ,0
Exp/Cntr=0,0

Type RM Length L Ch R = 1 ,265     ,5,5,5
#Sta/Elev= 4
 0.00000 4.81791 0.00000-0.18209  100000-0.18209  100000 4.81791
#Mann= 3 ,0,0
 0.00000 0.03000 0.00000 0.00000 0.03000 0.00000  100000 0.03000 0.00000
Bank Sta=0,100000
XS Rating Curve= 0 ,0
Exp/Cntr=0,0

Type RM Length L Ch R = 1 ,260     ,5,5,5
#Sta/Elev= 4
 0.00000 4.82333 0.00000-0.17667  100000-0.17667  100000 4.82333
#Mann= 3 ,0,0
 0.00000 0.03000 0.00000 0.00000 0.03000 0.00000  100000 0.03000 0.00000
Bank Sta=0,100000
XS Rating Curve= 0 ,0
Exp/Cntr=0,0

Type RM Length L Ch R = 1 ,255     ,5,5,5
#Sta/Elev= 4
 0.00000 4.82864 0.00000-0.17136  100000-0.17136  100000 4.82864
#Mann= 3 ,0,0
 0.00000 0.03000 0.00000 0.00000 0.03000 0.00000  100000 0.03000 0.00000
Bank Sta=0,100000
XS Rating Curve= 0 ,0
Exp/Cntr=0,0

Type RM Length L Ch R = 1 ,250     ,5,5,5
#Sta/Elev= 4
 0.00000 4.83384 0.00000-0.16616  100000-0.16616  100000 4.83384
#Mann= 3 ,0,0
 0.00000 0.03000 0.00000 0.00000 0.03000 0.00000  100000 0.03000 0.00000
Bank Sta=0,100000
XS Rating Curve= 0 ,0
Exp/Cntr=0,0

Type RM Length L Ch R = 1 ,245     ,5,5,5
#Sta/Elev= 4
 0.00000 4.83893 0.00000-0.16107  100000-0.16107  100000 4.83893
#Mann= 3 ,0,0
 0.00000 0.03000 0.00000 0.00000 0.03000 0.00000  100000 0.03000 0.00000
Bank Sta=0,100000
XS Rating Curve= 0 ,0
Exp/Cntr=0,0

Type RM Length L Ch R = 1 ,240     ,5,5,5
#Sta/Elev= 4
 0.00000  4.8439 0.00000-0.15610  100000-0.15610  100000  4.8439
#Mann= 3 ,0,0
 0.00000 0.03000 0.00000 0.00000 0.03000 0.00000  100000 0.03000 0.00000
Bank Sta=0,100000
XS Rating Curve= 0 ,0
Exp/Cntr=0,0

Type RM Length L Ch R = 1 ,235     ,5,5,5
#Sta/Elev= 4
 0.00000 4.84874 0.00000-0.15126  100000-0.15126  100000 4.84874
#Mann= 3 ,0,0
 0.00000 0.03000 0.00000 0.00000 0.03000 0.00000  100000 0.03000 0.00000
Bank Sta=0,100000
XS Rating Curve= 0 ,0
Exp/Cntr=0,0

Type RM Length L Ch R = 1 ,230     ,5,5,5
#Sta/Elev= 4
 0.00000 4.85346 0.00000-0.14654  100000-0.14654  100000 4.85346
#Mann= 3 ,0,0
 0.00000 0.03000 0.00000 0.00000 0.03000 0.00000  100000 0.03000 0.00000
Bank Sta=0,100000
XS Rating Curve= 0 ,0
Exp/Cntr=0,0

Type RM Length L Ch R = 1 ,225     ,5,5,5
#Sta/Elev= 4
 0.00000 4.85805 0.00000-0.14195  100000-0.14195  100000 4.85805
#Mann= 3 ,0,0
 0.00000 0.03000 0.00000 0.00000 0.03000 0.00000  100000 0.03000 0.00000
Bank Sta=0,100000
XS Rating Curve= 0 ,0
Exp/Cntr=0,0

Type RM Length L Ch R = 1 ,220     ,5,5,5
#Sta/Elev= 4
 0.00000 4.86251 0.00000-0.13749  100000-0.13749  100000 4.86251
#Mann= 3 ,0,0
 0.00000 0.03000 0.00000 0.00000 0.03000 0.00000  100000 0.03000 0.00000
Bank Sta=0,100000
XS Rating Curve= 0 ,0
Exp/Cntr=0,0

Type RM Length L Ch R = 1 ,215     ,5,5,5
#Sta/Elev= 4
 0.00000 4.86684 0.00000-0.13316  100000-0.13316  100000 4.86684
#Mann= 3 ,0,0
 0.00000 0.03000 0.00000 0.00000 0.03000 0.00000  100000 0.03000 0.00000
Bank Sta=0,100000
XS Rating Curve= 0 ,0
Exp/Cntr=0,0

Type RM Length L Ch R = 1 ,210     ,5,5,5
#Sta/Elev= 4
 0.00000 4.87103 0.00000-0.12897  100000-0.12897  100000 4.87103
#Mann= 3 ,0,0
 0.00000 0.03000 0.00000 0.00000 0.03000 0.00000  100000 0.03000 0.00000
Bank Sta=0,100000
XS Rating Curve= 0 ,0
Exp/Cntr=0,0

Type RM Length L Ch R = 1 ,205     ,5,5,5
#Sta/Elev= 4
 0.00000 4.87509 0.00000-0.12491  100000-0.12491  100000 4.87509
#Mann= 3 ,0,0
 0.00000 0.03000 0.00000 0.00000 0.03000 0.00000  100000 0.03000 0.00000
Bank Sta=0,100000
XS Rating Curve= 0 ,0
Exp/Cntr=0,0

Type RM Length L Ch R = 1 ,200     ,5,5,5
#Sta/Elev= 4
 0.00000 4.87901 0.00000-0.12099  100000-0.12099  100000 4.87901
#Mann= 3 ,0,0
 0.00000 0.03000 0.00000 0.00000 0.03000 0.00000  100000 0.03000 0.00000
Bank Sta=0,100000
XS Rating Curve= 0 ,0
Exp/Cntr=0,0

Type RM Length L Ch R = 1 ,195     ,5,5,5
#Sta/Elev= 4
 0.00000 4.88279 0.00000-0.11721  100000-0.11721  100000 4.88279
#Mann= 3 ,0,0
 0.00000 0.03000 0.00000 0.00000 0.03000 0.00000  100000 0.03000 0.00000
Bank Sta=0,100000
XS Rating Curve= 0 ,0
Exp/Cntr=0,0

Type RM Length L Ch R = 1 ,190     ,5,5,5
#Sta/Elev= 4
 0.00000 4.88643 0.00000-0.11357  100000-0.11357  100000 4.88643
#Mann= 3 ,0,0
 0.00000 0.03000 0.00000 0.00000 0.03000 0.00000  100000 0.03000 0.00000
Bank Sta=0,100000
XS Rating Curve= 0 ,0
Exp/Cntr=0,0

Type RM Length L Ch R = 1 ,185     ,5,5,5
#Sta/Elev= 4
 0.00000 4.88994 0.00000-0.11006  100000-0.11006  100000 4.88994
#Mann= 3 ,0,0
 0.00000 0.03000 0.00000 0.00000 0.03000 0.00000  100000 0.03000 0.00000
Bank Sta=0,100000
XS Rating Curve= 0 ,0
Exp/Cntr=0,0

Type RM Length L Ch R = 1 ,180     ,5,5,5
#Sta/Elev= 4
 0.00000 4.89331 0.00000-0.10669  100000-0.10669  100000 4.89331
#Mann= 3 ,0,0
 0.00000 0.03000 0.00000 0.00000 0.03000 0.00000  100000 0.03000 0.00000
Bank Sta=0,100000
XS Rating Curve= 0 ,0
Exp/Cntr=0,0

Type RM Length L Ch R = 1 ,175     ,5,5,5
#Sta/Elev= 4
 0.00000 4.89654 0.00000-0.10346  100000-0.10346  100000 4.89654
#Mann= 3 ,0,0
 0.00000 0.03000 0.00000 0.00000 0.03000 0.00000  100000 0.03000 0.00000
Bank Sta=0,100000
XS Rating Curve= 0 ,0
Exp/Cntr=0,0

Type RM Length L Ch R = 1 ,170     ,5,5,5
#Sta/Elev= 4
 0.00000 4.89964 0.00000-0.10036  100000-0.10036  100000 4.89964
#Mann= 3 ,0,0
 0.00000 0.03000 0.00000 0.00000 0.03000 0.00000  100000 0.03000 0.00000
Bank Sta=0,100000
XS Rating Curve= 0 ,0
Exp/Cntr=0,0

Type RM Length L Ch R = 1 ,165     ,5,5,5
#Sta/Elev= 4
 0.00000 4.90261 0.00000-0.09739  100000-0.09739  100000 4.90261
#Mann= 3 ,0,0
 0.00000 0.03000 0.00000 0.00000 0.03000 0.00000  100000 0.03000 0.00000
Bank Sta=0,100000
XS Rating Curve= 0 ,0
Exp/Cntr=0,0

Type RM Length L Ch R = 1 ,160     ,5,5,5
#Sta/Elev= 4
 0.00000 4.90544 0.00000-0.09456  100000-0.09456  100000 4.90544
#Mann= 3 ,0,0
 0.00000 0.03000 0.00000 0.00000 0.03000 0.00000  100000 0.03000 0.00000
Bank Sta=0,100000
XS Rating Curve= 0 ,0
Exp/Cntr=0,0

Type RM Length L Ch R = 1 ,155     ,5,5,5
#Sta/Elev= 4
 0.00000 4.90815 0.00000-0.09185  100000-0.09185  100000 4.90815
#Mann= 3 ,0,0
 0.00000 0.03000 0.00000 0.00000 0.03000 0.00000  100000 0.03000 0.00000
Bank Sta=0,100000
XS Rating Curve= 0 ,0
Exp/Cntr=0,0

Type RM Length L Ch R = 1 ,150     ,5,5,5
#Sta/Elev= 4
 0.00000 4.91072 0.00000-0.08928  100000-0.08928  100000 4.91072
#Mann= 3 ,0,0
 0.00000 0.03000 0.00000 0.00000 0.03000 0.00000  100000 0.03000 0.00000
Bank Sta=0,100000
XS Rating Curve= 0 ,0
Exp/Cntr=0,0

Type RM Length L Ch R = 1 ,145     ,5,5,5
#Sta/Elev= 4
 0.00000 4.91317 0.00000-0.08683  100000-0.08683  100000 4.91317
#Mann= 3 ,0,0
 0.00000 0.03000 0.00000 0.00000 0.03000 0.00000  100000 0.03000 0.00000
Bank Sta=0,100000
XS Rating Curve= 0 ,0
Exp/Cntr=0,0

Type RM Length L Ch R = 1 ,140     ,5,5,5
#Sta/Elev= 4
 0.00000  4.9155 0.00000-0.08450  100000-0.08450  100000  4.9155
#Mann= 3 ,0,0
 0.00000 0.03000 0.00000 0.00000 0.03000 0.00000  100000 0.03000 0.00000
Bank Sta=0,100000
XS Rating Curve= 0 ,0
Exp/Cntr=0,0

Type RM Length L Ch R = 1 ,135     ,5,5,5
#Sta/Elev= 4
 0.00000  4.9177 0.00000-0.08230  100000-0.08230  100000  4.9177
#Mann= 3 ,0,0
 0.00000 0.03000 0.00000 0.00000 0.03000 0.00000  100000 0.03000 0.00000
Bank Sta=0,100000
XS Rating Curve= 0 ,0
Exp/Cntr=0,0

Type RM Length L Ch R = 1 ,130     ,5,5,5
#Sta/Elev= 4
 0.00000 4.91979 0.00000-0.08021  100000-0.08021  100000 4.91979
#Mann= 3 ,0,0
 0.00000 0.03000 0.00000 0.00000 0.03000 0.00000  100000 0.03000 0.00000
Bank Sta=0,100000
XS Rating Curve= 0 ,0
Exp/Cntr=0,0

Type RM Length L Ch R = 1 ,125     ,5,5,5
#Sta/Elev= 4
 0.00000 4.92176 0.00000-0.07824  100000-0.07824  100000 4.92176
#Mann= 3 ,0,0
 0.00000 0.03000 0.00000 0.00000 0.03000 0.00000  100000 0.03000 0.00000
Bank Sta=0,100000
XS Rating Curve= 0 ,0
Exp/Cntr=0,0

Type RM Length L Ch R = 1 ,120     ,5,5,5
#Sta/Elev= 4
 0.00000 4.92362 0.00000-0.07638  100000-0.07638  100000 4.92362
#Mann= 3 ,0,0
 0.00000 0.03000 0.00000 0.00000 0.03000 0.00000  100000 0.03000 0.00000
Bank Sta=0,100000
XS Rating Curve= 0 ,0
Exp/Cntr=0,0

Type RM Length L Ch R = 1 ,115     ,5,5,5
#Sta/Elev= 4
 0.00000 4.92537 0.00000-0.07463  100000-0.07463  100000 4.92537
#Mann= 3 ,0,0
 0.00000 0.03000 0.00000 0.00000 0.03000 0.00000  100000 0.03000 0.00000
Bank Sta=0,100000
XS Rating Curve= 0 ,0
Exp/Cntr=0,0

Type RM Length L Ch R = 1 ,110     ,5,5,5
#Sta/Elev= 4
 0.00000 4.92701 0.00000-0.07299  100000-0.07299  100000 4.92701
#Mann= 3 ,0,0
 0.00000 0.03000 0.00000 0.00000 0.03000 0.00000  100000 0.03000 0.00000
Bank Sta=0,100000
XS Rating Curve= 0 ,0
Exp/Cntr=0,0

Type RM Length L Ch R = 1 ,105     ,5,5,5
#Sta/Elev= 4
 0.00000 4.92854 0.00000-0.07146  100000-0.07146  100000 4.92854
#Mann= 3 ,0,0
 0.00000 0.03000 0.00000 0.00000 0.03000 0.00000  100000 0.03000 0.00000
Bank Sta=0,100000
XS Rating Curve= 0 ,0
Exp/Cntr=0,0

Type RM Length L Ch R = 1 ,100     ,5,5,5
#Sta/Elev= 4
 0.00000 4.92998 0.00000-0.07002  100000-0.07002  100000 4.92998
#Mann= 3 ,0,0
 0.00000 0.03000 0.00000 0.00000 0.03000 0.00000  100000 0.03000 0.00000
Bank Sta=0,100000
XS Rating Curve= 0 ,0
Exp/Cntr=0,0

Type RM Length L Ch R = 1 ,95      ,5,5,5
#Sta/Elev= 4
 0.00000 4.93132 0.00000-0.06868  100000-0.06868  100000 4.93132
#Mann= 3 ,0,0
 0.00000 0.03000 0.00000 0.00000 0.03000 0.00000  100000 0.03000 0.00000
Bank Sta=0,100000
XS Rating Curve= 0 ,0
Exp/Cntr=0,0

Type RM Length L Ch R = 1 ,90      ,5,5,5
#Sta/Elev= 4
 0.00000 4.93257 0.00000-0.06743  100000-0.06743  100000 4.93257
#Mann= 3 ,0,0
 0.00000 0.03000 0.00000 0.00000 0.03000 0.00000  100000 0.03000 0.00000
Bank Sta=0,100000
XS Rating Curve= 0 ,0
Exp/Cntr=0,0

Type RM Length L Ch R = 1 ,85      ,5,5,5
#Sta/Elev= 4
 0.00000 4.93372 0.00000-0.06628  100000-0.06628  100000 4.93372
#Mann= 3 ,0,0
 0.00000 0.03000 0.00000 0.00000 0.03000 0.00000  100000 0.03000 0.00000
Bank Sta=0,100000
XS Rating Curve= 0 ,0
Exp/Cntr=0,0

Type RM Length L Ch R = 1 ,80      ,5,5,5
#Sta/Elev= 4
 0.00000 4.93479 0.00000-0.06521  100000-0.06521  100000 4.93479
#Mann= 3 ,0,0
 0.00000 0.03000 0.00000 0.00000 0.03000 0.00000  100000 0.03000 0.00000
Bank Sta=0,100000
XS Rating Curve= 0 ,0
Exp/Cntr=0,0

Type RM Length L Ch R = 1 ,75      ,5,5,5
#Sta/Elev= 4
 0.00000 4.93578 0.00000-0.06422  100000-0.06422  100000 4.93578
#Mann= 3 ,0,0
 0.00000 0.03000 0.00000 0.00000 0.03000 0.00000  100000 0.03000 0.00000
Bank Sta=0,100000
XS Rating Curve= 0 ,0
Exp/Cntr=0,0

Type RM Length L Ch R = 1 ,70      ,5,5,5
#Sta/Elev= 4
 0.00000 4.93668 0.00000-0.06332  100000-0.06332  100000 4.93668
#Mann= 3 ,0,0
 0.00000 0.03000 0.00000 0.00000 0.03000 0.00000  100000 0.03000 0.00000
Bank Sta=0,100000
XS Rating Curve= 0 ,0
Exp/Cntr=0,0

Type RM Length L Ch R = 1 ,65      ,5,5,5
#Sta/Elev= 4
 0.00000  4.9375 0.00000-0.06250  100000-0.06250  100000  4.9375
#Mann= 3 ,0,0
 0.00000 0.03000 0.00000 0.00000 0.03000 0.00000  100000 0.03000 0.00000
Bank Sta=0,100000
XS Rating Curve= 0 ,0
Exp/Cntr=0,0

Type RM Length L Ch R = 1 ,60      ,5,5,5
#Sta/Elev= 4
 0.00000 4.93826 0.00000-0.06174  100000-0.06174  100000 4.93826
#Mann= 3 ,0,0
 0.00000 0.03000 0.00000 0.00000 0.03000 0.00000  100000 0.03000 0.00000
Bank Sta=0,100000
XS Rating Curve= 0 ,0
Exp/Cntr=0,0
